HEC-RAS study SFSBPOTOMC.prj: SFSBPOTOMC

--- SFSBPOTOMC.g01 (geometry) --- (continued)

Type RM Length L Ch R = 1 ,45988   ,683.7,678.7,671.6
XS GIS Cut Line= 4
2487367.59498726627585.3339240792487581.67963873626949.376577058
2487783.17107541626596.766562868 2488305.7894893625576.716164676
#Sta/Elev= 30
       0 1528.41    74.3 1502.57   133.4 1484.96   154.5  1480.4  215.96 1474.79
   283.71467.901  325.851467.206   487.5 1458.52   561.5 1451.37   745.7 1442.11
   790.9 1429.23  824.691424.782   834.9 1419.96     907 1419.68   977.9 1424.68
   995.7  1427.3 1027.671426.806  1339.4 1427.57  1434.8 1423.98  1538.9 1428.65
    1650 1429.86 1849.731427.219  1870.3 1427.68  1892.7 1434.47  1951.2 1472.23
  1996.1 1488.96  2063.5 1500.32 2113.751501.157  2180.4 1499.36  2223.3 1510.97
#Mann= 9 ,-1 , 0
       0      .1       0  215.96      .1       0   283.7      .1       0
  325.85      .1       0  824.69    .045       0   977.9     .12       0
 1027.67     .05       0 1849.73      .1       0 2113.75     .05       0
Bank Sta=824.69,977.9
XS Rating Curve= 0 ,0
Exp/Cntr(USF)=0,0
Exp/Cntr=0.3,0.1

Type RM Length L Ch R = 1 ,45309   ,557,600.6,636.7
XS GIS Cut Line= 4
2487921.69643813627786.8253607592488160.96751919627346.062843022
2488375.05217066626892.7071104922488740.25539964626042.665111999
#Sta/Elev= 30
       0 1458.13     4.5 1454.88    13.6 1453.11    35.7  1457.1    94.4 1455.19
   133.5 1461.57  186.791460.231   241.1 1459.73   286.7 1464.22   372.4 1481.31
   428.5 1482.82     455 1481.23   496.3 1475.69   580.4 1456.55   637.7  1439.6
   664.3  1426.6  687.771423.585  712.271421.332   748.6 1419.32   787.7 1416.39
   876.6 1418.88  947.861424.032  1261.7 1430.75  1366.2 1439.52    1475 1439.59
  1713.6 1445.52  1759.2 1452.84  1823.3 1473.32 1869.961484.861  1928.1 1493.97
#Mann= 8 ,-1 , 0
       0      .1       0  186.79      .1       0  687.77      .1       0
  712.27    .025       0   748.6    .045       0   876.6      .1       0
  947.86     .05       0 1869.96      .1       0
Bank Sta=748.6,876.6
XS Rating Curve= 0 ,0
Exp/Cntr(USF)=0,0
Exp/Cntr=0.3,0.1

Type RM Length L Ch R = 1 ,44708   ,572.6,576.2,574.3
XS GIS Cut Line= 4
2488261.71323753627780.5287533632488400.23860024627686.079642419
2488916.56040674627402.7323095882490748.87315905626710.105496001
#Sta/Elev= 30
       0 1537.58    39.3 1538.25      81 1532.22   140.1 1515.44  192.07 1494.45
     239  1472.6  297.461439.322  321.521422.421   333.9 1415.75   348.5 1414.84
   421.5  1416.6  457.471422.423  613.631425.897  628.431426.824  719.021429.542
  923.161431.904 1024.511436.042 1125.861437.934 1328.561440.973 1491.841444.536
  1635.6 1445.62  1686.9 1455.39  1763.9 1452.83 1835.311459.022 2038.011465.355
  2240.71469.317  2375.4 1472.08  2448.1 1478.79  2631.9 1532.88  2715.5 1548.54
#Mann= 16 ,-1 , 0
       0      .1       0  192.07    .025       0  297.46     .05       0
  321.52    .045       0  457.47      .1       0  613.63     .05       0
  628.43      .1       0  719.02     .05       0  923.16      .1       0
 1024.51     .05       0 1125.86      .1       0 1328.56     .05       0
 1491.84      .1       0 1835.31     .05       0 2038.01     .06       0
  2240.7      .1       0
Bank Sta=321.52,457.47
XS Rating Curve= 0 ,0
Exp/Cntr(USF)=0,0
Exp/Cntr=0.3,0.1

Type RM Length L Ch R = 1 ,44132   ,582.6,564.2,554.8
XS GIS Cut Line= 4
2488526.17074817628284.2573450632488715.06897006628164.621804534
2489445.47542802627774.2321459672490622.94101112627125.681584153
#Sta/Elev= 30
       0 1583.56    85.9 1556.71   160.8 1525.87  209.941502.162   260.1 1473.85
  315.311435.691  338.241421.045   350.2 1414.86   454.5    1416  465.531421.044
  505.151424.413  525.271424.386   617.8    1423   658.6 1430.44  735.241432.696
  800.281436.039  840.23 1436.99 1261.081446.326  1834.1 1458.01 1893.77 1464.52
 1948.571473.209 1999.221478.563  2044.2 1481.47  2080.7 1479.43 2104.67 1485.16
 2210.111491.142 2233.461494.878  2285.8 1505.64  2313.6 1505.64    2396 1526.98
#Mann= 17 ,-1 , 0
       0      .1       0  209.94    .025       0  315.31      .1       0
  338.24    .045       0  465.53    .025       0  505.15    .055       0
  525.27     .05       0  735.24     .05       0  800.28     .05       0
  840.23     .05       0 1261.08     .05       0 1893.77      .1       0
 1948.57     .05       0 1999.22     .06       0 2104.67     .12       0
 2210.11      .1       0 2233.46     .12       0
Bank Sta=338.24,465.53
XS Rating Curve= 0 ,0
Exp/Cntr(USF)=0,0
Exp/Cntr=0.3,0.1

Type RM Length L Ch R = 1 ,43568   ,729.3,658.8,629.2
XS GIS Cut Line= 4
  2488809.518081628850.9520107252488960.63665851628731.316470196
2489363.61953187628403.8928855912490358.48350048627471.994990947
#Sta/Elev= 30
       0 1610.07    4.641608.699   11.09 1607.27  118.361577.508   180.3 1548.57
   217.3 1526.48   262.5 1493.29   282.2 1475.05   294.1 1467.06   322.5 1440.14
  346.921431.214   386.2 1422.41  391.76 1419.14   396.4 1415.13   402.7 1414.69
   524.4 1414.76  542.441419.141  576.011419.643   615.4  1423.3  690.561423.751
   789.5 1433.31 1048.651437.383 1407.691444.438 1473.191446.743  1552.6 1451.02
 1647.061461.245  1835.5 1472.68  2006.11488.029  2053.5 1492.27  2075.1 1496.83
#Mann= 14 ,-1 , 0
       0      .1       0    4.64      .1       0   11.09      .1       0
  118.36      .1       0  346.92    .025       0  391.76    .045       0
  542.44    .025       0  576.01      .1       0  690.56     .05       0
 1048.65     .05       0 1407.69      .1       0 1473.19     .05       0
 1647.06      .1       0  2006.1     .06       0
Bank Sta=391.76,542.44
XS Rating Curve= 0 ,0
Exp/Cntr(USF)=0,0
Exp/Cntr=0.3,0.1

Type RM Length L Ch R = 1 ,42909   ,711.9,753.9,795.1
XS GIS Cut Line= 4
2489124.34845081629512.0957873312489760.30579783628920.214692084
2489854.75490878628561.3080704982490629.23761852627679.783035023
#Sta/Elev= 30
       0 1640.64    52.5 1628.68   107.3 1605.57   154.4 1577.66   210.9 1531.28
   240.3 1513.05   254.2 1498.21   318.8 1458.76   376.1 1430.61   413.1 1426.11
   440.4 1415.15   475.2 1411.61   540.3 1420.36   664.5 1422.57   857.3 1421.66
   903.2 1416.15   998.4 1421.92  1022.5 1417.47  1039.7 1411.18  1061.8 1410.47
  1105.9  1410.7 1117.171416.906  1134.9 1430.47 1214.981431.705 1812.83 1443.67
  1967.2 1456.34 2164.571481.857    2245  1491.8 2293.261503.989  2413.3 1525.22
#Mann= 7 ,-1 , 0
       0      .1       0  1022.5    .045       0 1117.17      .1       0
 1214.98     .05       0 1812.83      .1       0 2164.57     .06       0
 2293.26      .1       0
Bank Sta=1022.5,1117.17
XS Rating Curve= 0 ,0
Exp/Cntr(USF)=0,0
Exp/Cntr=0.3,0.1

Type RM Length L Ch R = 1 ,42155   ,312.7,316.2,320
XS GIS Cut Line= 4
2489262.87381353629650.6211500482490383.66993006629014.663803027
2490648.12744071628838.3587959322491183.33906939628378.706456006
#Sta/Elev= 30
       0 1630.05    73.1 1590.65     124 1538.46   142.4 1529.77   160.8  1507.3
     252 1454.21   317.2 1429.07   413.8 1408.09   473.6 1417.69   542.5 1420.69
   583.9 1416.38   781.7 1418.92   841.8 1415.61 1065.881415.298 1146.57 1417.63
  1368.6  1413.8    1409 1408.88  1465.4 1410.01 1477.091414.223  1494.3 1428.53
  1508.7 1434.61  1578.81440.629  1725.9 1458.32  1837.7 1463.41  1931.6 1462.33
 2042.611474.651  2073.2 1477.54 2159.021518.784  2268.9 1566.06    2312 1577.38
#Mann= 8 ,-1 , 0
       0      .1       0 1065.88      .1       0 1146.57      .1       0
  1368.6    .045       0 1477.09      .1       0  1578.8     .05       0
 2042.61     .06       0 2159.02      .1       0
Bank Sta=1368.6,1477.09
XS Rating Curve= 0 ,0
Exp/Cntr(USF)=0,0
Exp/Cntr=0.3,0.1

Type RM Length L Ch R = 1 ,41839   ,560.7,565.7,571.3
XS GIS Cut Line= 4
2489388.80596146629889.8922311062490452.93261142 629329.49417284
 2490824.4324478629115.409521367 2491334.4576469628750.206292385
#Sta/Elev= 30
       0 1628.62    24.4 1612.25    83.7  1563.4   110.7 1534.76   169.5 1479.33
   240.6 1442.03     278 1429.77   332.4 1424.33   382.7 1410.16   486.3 1416.05
   766.2 1412.91  938.421415.702 1147.951413.662  1261.5 1416.17    1371    1413
  1384.8 1407.75  1425.6 1407.13  1466.6 1407.34 1493.081412.815  1541.8  1431.6
 1605.741435.404  1791.7 1443.41  1973.7 1463.73 2043.841466.919  2112.2 1474.04
  2149.5  1470.7  2185.3 1487.76  2198.2 1497.04 2234.641508.081  2258.7  1517.1
#Mann= 8 ,-1 , 0
       0      .1       0  938.42     .05       0 1147.95      .1       0
    1371    .045       0 1493.08      .1       0 1605.74     .05       0
 2043.84     .06       0 2234.64      .1       0
Bank Sta=1371,1493.08
XS Rating Curve= 0 ,0
Exp/Cntr(USF)=0,0
Exp/Cntr=0.3,0.1

Type RM Length L Ch R = 1 ,41273   ,376.8,373.6,370.5
XS GIS Cut Line= 4
2489502.14489459630425.1038597872490774.05958863 629782.84990537
2491145.55942501629606.5448982752491548.54229837 629379.86703201
#Sta/Elev= 30
       0 1694.47   72.221663.419     151 1615.31   233.7 1544.23  280.591516.008
   341.2 1473.36   395.1 1443.48   502.5 1413.39     525 1410.86   547.4 1414.12
   762.4 1412.12   794.1 1406.34   829.7 1405.81   892.3 1415.03 1009.861414.373
  1304.7  1410.6  1456.6  1414.4  1515.4 1410.07  1530.4  1406.7  1629.5 1406.62
 1646.66 1410.49 1736.811419.046 1840.311428.101    1869 1432.65  1901.7  1448.8
  1946.11454.478  2039.4 1463.66  2115.7 1466.72 2221.521483.286  2298.4 1501.44
#Mann= 10 ,-1 , 0
       0      .1       0   72.22      .1       0  280.59      .1       0
 1009.86     .05       0  1515.4    .045       0 1646.66      .1       0
 1736.81      .1       0 1840.31     .06       0  1946.1      .1       0
 2221.52      .1       0
Bank Sta=1515.4,1646.66
XS Rating Curve= 0 ,0
Exp/Cntr(USF)=0,0
Exp/Cntr=0.3,0.1

Type RM Length L Ch R = 1 ,40900   ,554.7,540.1,522.8
XS GIS Cut Line= 4
2489672.15329429630891.0528071092490767.76298123630217.315815711
2491265.19496554629952.8583050682491529.65247618629663.214364841
#Sta/Elev= 30
       0 1745.39   81.02 1710.51   143.9 1674.11   247.2 1598.98   284.1 1567.53
   472.6 1446.82   505.5 1433.05   594.7  1418.8   641.7 1402.75   777.8 1409.59
   970.4 1408.12  1007.9  1413.8 1047.661413.576  1237.4 1409.35  1458.8 1411.08
 1472.831407.642  1488.4  1404.9  1525.1 1409.59 1577.16 1409.43  1594.8 1407.63
    1722 1408.79  1869.6 1410.46 1901.38 1417.79  1946.8 1424.27  1964.6 1444.13
 2028.091489.683  2047.2 1497.74  2083.2 1504.59 2173.921508.729  2241.8 1508.49
#Mann= 10 ,-1 , 0
       0      .1       0   81.02      .1       0 1047.66     .05       0
 1472.83      .1       0 1577.16    .025       0  1594.8    .045       0
    1722      .1       0 1901.38     .06       0 2028.09      .1       0
 2173.92      .1       0
Bank Sta=1594.8,1722
XS Rating Curve= 0 ,0
Exp/Cntr(USF)=0,0
Exp/Cntr=0.3,0.1

Type RM Length L Ch R = 1 ,40360   ,419.9,433.9,445.4
XS GIS Cut Line= 4
 2489986.9836641631363.2983618282491410.01693565630475.476718957
2491611.50837233630305.4683192582491869.66927558630122.866704767
#Sta/Elev= 30
       0 1744.46   41.581730.382   108.2  1697.9   235.5 1607.25   329.7 1512.07
   409.9 1463.11   508.9 1422.16   593.8 1401.05   630.1 1399.17   655.1  1405.5
   683.3 1402.34  795.441408.971  834.59 1408.24 1226.221408.077 1333.911407.785
 1441.611409.893  1503.7 1409.54  1518.5  1403.4  1549.31401.831 1579.35 1407.61
 1656.991408.665    1734 1405.08  1831.5 1405.08 1887.071406.008  1916.6 1411.45
 2000.061413.461  2028.2 1426.01 2110.621489.547  2180.9  1501.2  2257.1 1503.14
#Mann= 15 ,-1 , 0
       0      .1       0   41.58      .1       0  795.44     .05       0
  834.59      .1       0 1226.22     .05       0 1333.91      .1       0
 1441.61      .1       0  1549.3      .1       0 1579.35      .1       0
 1656.99      .1       0    1734    .045       0  1831.5      .1       0
 1887.07     .06       0 2000.06      .1       0 2110.62      .1       0
Bank Sta=1734,1831.5
XS Rating Curve= 0 ,0
Exp/Cntr(USF)=0,0
Exp/Cntr=0.3,0.1

Type RM Length L Ch R = 1 ,39926   ,383,385.2,386.5
XS GIS Cut Line= 4
2490276.62760433 631678.128731642491441.49997263630897.349414505
2491844.48284599630702.154585222 2492165.6098232630551.036007712
#Sta/Elev= 30
       0 1720.35   142.3 1630.33   199.8 1588.76   262.6 1539.17   300.8 1500.53
  329.351477.903   395.9 1440.89   438.61424.302   463.11418.576   580.4 1397.75
   657.11405.073  693.831406.241   875.61405.738   980.1 1401.06  1094.11408.854
  1211.2  1408.8  1273.8 1403.25  1312.61406.264  1492.6 1401.82  1643.7 1404.26
  1661.5 1400.29 1722.221404.052 1731.811406.572  1768.2 1411.08 1835.461409.638
 1938.821415.172  2028.6  1475.2  2047.1 1483.04  2094.7 1489.53    2205  1492.8
#Mann= 14 ,-1 , 0
       0      .1       0  329.35     .05       0   438.6      .1       0
   463.1     .05       0   657.1      .1       0  693.83     .05       0
   875.6      .1       0  1094.1     .05       0  1312.6      .1       0
  1643.7    .045       0 1722.22      .1       0 1731.81     .06       0
 1835.46      .1       0 1938.82      .1       0
Bank Sta=1643.7,1722.22
XS Rating Curve= 0 ,0
Exp/Cntr(USF)=0,0
Exp/Cntr=0.3,0.1

Type RM Length L Ch R = 1 ,39540   ,485.3,507.5,526.7
XS GIS Cut Line= 4
2490408.85635965631759.9846277912491592.61855014631237.366213903
 2492001.8980309631061.0612068082492310.43179331630960.315488468
#Sta/Elev= 30
       0 1689.68    56.9 1658.54      72 1635.29   102.6 1611.87   153.9 1585.31
   178.2 1563.25   238.2 1529.78     254 1515.34   299.4 1486.04  393.731435.095
   507.8 1407.26   678.7 1395.63  701.231402.221   906.51404.886 1111.771404.055
  1125.8 1399.59    1152 1399.04    1257 1400.14  1291.9 1405.61  1527.1 1405.53
  1544.6 1401.66 1615.37 1402.71 1624.181406.423 1726.581409.028 1827.341412.237
  1849.9 1421.17  1938.3 1488.73  1963.5 1495.94 2028.371504.151  2064.2 1513.77
#Mann= 11 ,-1 , 0
       0      .1       0  393.73     .05       0  701.23      .1       0
   906.5     .05       0 1111.77      .1       0  1544.6    .045       0
 1615.37      .1       0 1624.18     .06       0 1726.58      .1       0
 1827.34      .1       0 2028.37     .12       0
Bank Sta=1544.6,1615.37
XS Rating Curve= 0 ,0
Exp/Cntr(USF)=0,0
Exp/Cntr=0.3,0.1

Type RM Length L Ch R = 1 ,39033   ,764.5,714.1,694.8
XS GIS Cut Line= 4
2490547.38172237 631879.620168322491454.09318743631508.120331941
2492014.49124569 631627.755872472492278.94875633631703.315161225
#Sta/Elev= 30
       0 1661.34    55.3 1632.13    92.1 1607.75   111.7 1589.11   163.6 1560.63
   223.9 1512.25   242.3 1501.95   331.2 1468.49  473.921423.712   550.5 1403.37
   634.8  1401.6  677.831395.045   682.3 1394.86   777.4 1402.77     812 1396.52
   876.8 1400.84   976.2 1398.26   996.9 1403.67  1258.7 1402.22  1315.9 1407.01
  1329.9 1400.11  1356.9 1396.35  1373.7 1400.07 1489.781399.252  1504.1 1404.33
 1625.361409.826  1668.9 1432.95    17321480.877  1775.8 1513.78  1827.9 1531.57
#Mann= 8 ,-1 , 0
       0      .1       0  473.92     .05       0  677.83      .1       0
  1329.9    .045       0  1373.7      .1       0 1489.78     .06       0
 1625.36      .1       0    1732      .1       0
Bank Sta=1329.9,1373.7
XS Rating Curve= 0 ,0
Exp/Cntr(USF)=0,0
Exp/Cntr=0.3,0.1

Type RM Length L Ch R = 1 ,38319   ,355.6,324.5,308.2
XS GIS Cut Line= 4
2490610.34779633631955.1794570752491044.81370667631942.586242282
2491517.05926139632062.221782811 2491661.8812315632225.933575114
#Sta/Elev= 30
       0 1654.46    64.4 1622.63   120.4  1584.8   160.5  1570.3     202 1546.48
   257.3 1520.85   316.5 1498.32   416.3 1472.94   486.2 1461.18   519.2 1450.11
   527.4  1442.6   539.8 1424.96   543.9 1422.24   560.4 1417.79   568.7 1418.04
   576.9 1413.19   638.8 1396.48  655.351394.018   684.2 1391.16   752.6 1390.11
   779.1 1390.58  797.921394.018   824.5 1395.29   849.3 1401.85   869.9 1413.65
   890.5 1451.82   894.7 1455.53  939.21 1465.56  1040.2 1477.15  1140.4 1479.25
#Mann= 4 ,-1 , 0
       0      .1       0  655.35    .045       0  797.92      .1       0
  939.21      .1       0
Bank Sta=655.35,797.92
XS Rating Curve= 0 ,0
Exp/Cntr(USF)=0,0
Exp/Cntr=0.3,0.1

Type RM Length L Ch R = 1 ,37994   ,238.2,216.1,199.6
XS GIS Cut Line= 4
2490742.57655165632427.4250117942491095.18656584632364.458937831
2491510.76265399 632332.97590085 2491661.8812315632288.899649076
#Sta/Elev= 30
       0 1700.89    65.2 1683.02    69.6 1679.58    77.4 1669.21    81.4 1666.67
    93.6 1663.72   109.9 1654.14   150.5 1635.36   176.4 1618.05   203.3 1604.15
   227.7 1583.26   292.7 1513.02   307.4 1499.13   369.8 1455.21   409.9 1430.94
     454 1413.02   510.2 1397.39  545.751392.379   566.3 1387.43     624 1386.58
   662.6 1387.64  680.37 1392.38   722.8 1409.21   730.8 1416.76   739.6 1422.14
   750.9 1435.67   765.7 1444.85   791.6 1456.06   862.4 1477.48   932.4 1481.85
#Mann= 3 ,-1 , 0
       0      .1       0  545.75    .045       0  680.37      .1       0
Bank Sta=545.75,680.37
XS Rating Curve= 0 ,0
Exp/Cntr(USF)=0,0
Exp/Cntr=0.3,0.1

Type RM Length L Ch R = 1 ,37778   ,320,311.1,317.8
XS GIS Cut Line= 4
2490969.25441791632710.7723446252491240.00853595632616.323233681
2491617.80497973632477.7978709632491762.62694984632402.238582209
#Sta/Elev= 30
       0 1657.23    51.3 1637.91    56.7 1630.71    65.1 1614.74    69.4 1610.63
   103.3 1589.46   145.6 1557.45   183.2 1532.83   217.6 1502.42   276.9 1461.63
   315.2 1437.08   323.8 1433.98   332.3 1425.08   346.1 1415.68   357.8 1411.49
   383.5 1409.82   400.4 1400.76   411.6 1398.87  427.66 1390.99   438.8 1386.68
   473.9 1386.34   528.3 1388.52   558.2 1389.01     608 1398.81   626.7 1409.18
   639.1  1424.2   647.5 1429.82   771.4 1472.94   825.4 1480.19   852.5 1481.15
#Mann= 3 ,-1 , 0
       0      .1       0  427.66    .045       0   528.3      .1       0
Bank Sta=427.66,528.3
XS Rating Curve= 0 ,0
Exp/Cntr(USF)=0,0
Exp/Cntr=0.3,0.1

Type RM Length L Ch R = 1 ,37467   ,315,307.9,304.3
XS GIS Cut Line= 4
2491076.29674365633031.8993218332491403.72032826632912.263781304
2491800.40659422632698.1791298322491863.37266818632572.246981907
#Sta/Elev= 30
       0 1670.57    36.7 1661.51    99.4 1639.63   117.6 1619.61   168.7 1596.42
   183.6 1584.79   224.1 1559.75   267.8 1528.95   287.9 1511.72   305.2 1489.07
   320.8 1475.12   334.8 1466.48   345.8 1450.17   370.2 1423.25   407.9 1404.79
   438.4 1393.23   454.31389.766   465.7 1385.45   529.3 1387.08   642.9 1385.93
   661.8 1386.65  673.281389.766     680 1392.16   694.3 1403.44   722.1 1417.04
   772.6 1446.54   825.4 1465.09   849.3 1470.24   872.1 1472.18   940.2 1473.76
#Mann= 3 ,-1 , 0
       0      .1       0   454.3    .045       0  673.28      .1       0
Bank Sta=454.3,673.28
XS Rating Curve= 0 ,0
Exp/Cntr(USF)=0,0
Exp/Cntr=0.3,0.1

Type RM Length L Ch R = 1 ,37159   ,535.2,555.3,576
XS GIS Cut Line= 4
2491252.60175075633378.2127286272491523.35586878633227.094151117
2491857.07606079632994.1196774562492108.94035664632591.136804096
#Sta/Elev= 30
       0 1646.37    5.681645.245    56.1 1632.77  111.341608.775   185.7 1570.96
   242.2 1536.06   309.4 1485.82   343.5 1454.15     402 1408.96   413.2 1402.02
   426.4 1396.11   444.8 1391.09  494.421387.719   504.5 1384.73     583  1384.2
   606.9  1384.7   621.5 1388.02   686.1 1384.07   749.7 1390.04   777.5 1403.26
  823.551430.699   867.1 1446.21   891.9 1452.52   942.6 1454.56   973.2 1451.83
  1032.2 1455.84 1082.871462.806  1093.5 1466.26  1144.4 1474.79  1192.3 1478.64
#Mann= 7 ,-1 , 0
       0     .12       0    5.68      .1       0  111.34      .1       0
  494.42    .045       0   621.5      .1       0  823.55     .06       0
 1082.87     .05       0
Bank Sta=494.42,621.5
XS Rating Curve= 0 ,0
Exp/Cntr(USF)=0,0
Exp/Cntr=0.3,0.1

Type RM Length L Ch R = 1 ,36604   ,461.6,465.8,470.8
XS GIS Cut Line= 4
2491435.20336524633762.3057797982491812.99980901633636.373631873
2492247.46571935633504.1448765522492921.20271075633170.424684551
#Sta/Elev= 30
       0 1608.28    97.2    1565   138.7  1542.8   235.6 1479.41   298.9 1433.76
     347 1407.17     421 1385.06  465.481380.707   508.8  1376.3   567.3 1376.59
   578.31380.708   588.2 1385.87     630  1388.3   692.7  1385.2   772.7 1389.32
   834.9 1384.23  890.671384.756   905.1 1380.99   927.3 1381.11   954.2 1391.37
  994.611392.939  1043.8 1392.32 1098.541398.332 1202.471409.451  1321.4 1427.19
  1378.3 1447.73 1410.331455.795  1440.9 1462.85  1485.4 1467.18  1604.2 1465.64
#Mann= 8 ,-1 , 0
       0      .1       0  465.48    .045       0   578.3      .1       0
  890.67     .06       0  994.61      .1       0 1098.54     .05       0
 1202.47      .1       0 1410.33     .05       0
Bank Sta=465.48,578.3
XS Rating Curve= 0 ,0
Exp/Cntr(USF)=0,0
Exp/Cntr=0.3,0.1

Type RM Length L Ch R = 1 ,36138   ,494.3,492.3,489
XS GIS Cut Line= 4
2491472.98300961634184.1784753472491875.96588297634089.729364403
2492385.99108207 633976.390431272493399.74487287633510.441483948
#Sta/Elev= 30
       0 1604.91    63.4 1585.22   129.2 1557.28   157.9 1543.15   219.6 1508.02
   293.5 1461.39   326.4 1434.64   355.1 1417.14   379.8 1408.88   465.5 1400.57
   527.4 1376.85   547.9 1374.32   617.5 1374.06   629.8 1375.56   662.6  1373.4
   687.2 1373.81   711.8 1378.68  812.28 1381.69   842.9 1385.92 1013.931387.536
  1227.6 1389.41 1323.091392.791 1510.931402.944  1696.6  1414.5  1715.8    1422
  1742.8 1422.84  1782.6 1417.98 1838.341418.993  1866.1 1420.35  2052.1 1446.28
#Mann= 8 ,-1 , 0
       0      .1       0   527.4    .045       0   629.8      .1       0
  812.28     .06       0 1013.93     .05       0 1323.09      .1       0
 1510.93     .05       0 1838.34      .1       0
Bank Sta=527.4,629.8
XS Rating Curve= 0 ,0
Exp/Cntr(USF)=0,0
Exp/Cntr=0.3,0.1

Type RM Length L Ch R = 1 ,35646   ,814.4,801.1,789.5
XS GIS Cut Line= 4
 2491498.1694392634713.0934966312491945.22856433634587.161348706
2492480.44019301634442.3393785932493664.20238351633970.093823874
#Sta/Elev= 30
       0    1598    57.4  1590.3   137.7 1573.71  176.331558.136   216.7  1540.8
  276.291506.749     412 1412.78   457.7 1388.96  476.211385.605  557.031385.987
  576.061385.338   619.4 1382.08  633.741376.111   656.6 1370.78   721.9 1370.62
  755.131376.112  775.761380.021   801.7 1382.77     810 1385.47  875.611384.722
  1262.6 1382.85 1686.831393.492 1788.581395.969  1869.8    1398  2103.9 1414.14
  2141.1 1418.16 2195.551429.583  2214.3 1434.49  2270.1 1455.53  2293.4  1460.7
#Mann= 13 ,-1 , 0
       0     .05       0  176.33      .1       0  276.29      .1       0
  476.21     .05       0  557.03      .1       0  576.06     .05       0
  633.74    .045       0  755.13      .1       0  775.76     .06       0
  875.61     .05       0 1686.83      .1       0 1788.58     .05       0
 2195.55      .1       0
Bank Sta=633.74,755.13
XS Rating Curve= 0 ,0
Exp/Cntr(USF)=0,0
Exp/Cntr=0.5,0.3

Type RM Length L Ch R = 1 ,34845   ,88.4,90.3,92.6
XS GIS Cut Line= 4
2491650.58369079635494.0545768742492112.19618666635419.286385462
2492595.07480028635204.4106366192493948.84539044634549.563467413
#Sta/Elev= 30
       0 1482.12    77.2  1468.3   129.8 1454.67   162.2 1442.75     219 1412.65
   267.6 1400.88   340.5    1394   517.8  1384.6   549.71385.513   685.71373.604
   715.6 1367.87   766.8 1367.73   822.8 1368.32  841.261373.605  857.841379.876
   873.2 1385.35   895.1 1386.57  960.551379.639  1026.9 1384.18  1109.9 1381.86
  1183.4 1384.18  1506.8 1381.44  1622.3  1377.5  1675.6 1387.55    2000 1401.56
  2218.9 1420.66  2284.8 1421.28 2411.151439.238 2458.341449.4052499.993 1456.56
#Mann= 8 ,-1 , 0
       0     .05       0   549.7     .06       0   685.7    .045       0
  841.26    .025       0  857.84    .055       0  960.55     .05       0
 2411.15      .1       0 2458.34      .1       0
Bank Sta=685.7,841.26
XS Rating Curve= 0 ,0
Exp/Cntr(USF)=0,0
Exp/Cntr=0.5,0.3

Type RM Length L Ch R = 1 ,34755   ,640.7,644.9,648.3
XS GIS Cut Line= 4
2491737.19618669635856.7863854622492212.89063111635467.897496581
2492667.75174224635276.9252743422493969.83507559634627.619718805
#Sta/Elev= 30
       0 1446.61      33 1445.75  123.231431.577     312 1413.13   337.8 1407.69
  485.511396.439  508.251394.898  703.971381.206   737.9 1378.55  761.371373.294
   785.6 1367.83   825.4 1367.44   885.4 1368.19  901.891373.292   908.31374.389
   933.1 1383.35 1010.471380.811  1047.4 1378.45  1084.1 1383.67  1246.8 1383.74
  1335.2 1379.75  1473.1 1381.18  1728.9 1377.08  1759.2 1384.75  2067.6 1400.63
    2224 1418.27    2385 1430.07 2466.08 1438.91  2519.1 1446.132562.749  1456.2
#Mann= 10 ,-1 , 0
       0      .1       0  123.23     .05       0  485.51     .06       0
  508.25    .055       0  703.97     .05       0  761.37    .045       0
  901.89     .06       0   908.3    .055       0 1010.47     .05       0
 2466.08      .1       0
Bank Sta=761.37,901.89
XS Rating Curve= 0 ,0
Exp/Cntr(USF)=0,0
Exp/Cntr=0.5,0.3

Type RM Length L Ch R = 1 ,34110   ,860.8,857.5,854.6
XS GIS Cut Line= 4
2491731.14391286636287.2453456932492417.47411905636066.864086824
2492870.82985158635903.1522945222494388.31223408635317.567806671
#Sta/Elev= 30
       0 1600.78   98.931544.335     218 1473.24   323.1 1416.11  400.261406.928
   470.1 1403.76   500.7 1398.88  601.141383.252  701.581380.619  802.521378.573
   849.9 1378.18  863.211371.451   892.3 1367.23   960.4  1366.4  1015.6 1367.22
  1030.11371.452  1041.2 1376.86  1065.5 1379.95 1105.681377.813  1279.9 1377.86
  1352.8 1372.82  1549.5 1378.74    1748 1376.12  1854.5 1378.49  2001.2 1374.56
  2038.8 1381.31  2394.7 1398.38 2526.161411.892 2530.031412.547  2829.4 1456.05
#Mann= 12 ,-1 , 0
       0      .1       0   98.93      .1       0  400.26     .05       0
   500.7     .06       0  601.14     .05       0  701.58    .025       0
  802.52     .05       0  863.21    .045       0  1030.1     .06       0
 1105.68     .05       0 2526.16      .1       0 2530.03      .1       0
Bank Sta=863.21,1030.1
XS Rating Curve= 0 ,0
Exp/Cntr(USF)=0,0
Exp/Cntr=0.3,0.1

Type RM Length L Ch R = 1 ,33252   ,624.2,625.3,626.4
XS GIS Cut Line= 4
2491901.15231256637175.0669885642492732.30448886636872.829833544
2493393.44826547636602.0757155052494766.10867785636029.084442447
#Sta/Elev= 30
       0 1534.67    31.5 1525.16    91.1 1497.31   107.5 1493.63   163.7  1469.2
  275.571408.626   299.6 1405.03   316.6 1397.98  376.671392.488   465.6 1384.11
   503.9 1374.22  578.861373.678  984.091375.526  1007.4 1368.06    1035    1366
    1081 1362.35  1142.1 1362.68    1155 1368.17 1187.991372.847 1289.951373.354
  1634.9 1375.31  2172.4 1369.06 2208.491372.645  2432.5 1372.62  2484.5 1383.61
  2728.6 1399.67  2857.2 1413.16 2923.291434.347  3025.41455.807  3086.3 1478.71
#Mann= 12 ,-1 , 0
       0      .1       0  275.57     .06       0  376.67     .05       0
  578.86     .05       0  984.09    .025       0    1035    .045       0
    1155      .1       0 1187.99     .06       0 1289.95     .05       0
 2208.49     .05       0 2923.29      .1       0  3025.4      .1       0
Bank Sta=1035,1155
XS Rating Curve= 0 ,0
Exp/Cntr(USF)=0,0
Exp/Cntr=0.3,0.1

Type RM Length L Ch R = 1 ,32627   ,631.3,610.8,581.9
XS GIS Cut Line= 4
 2492159.3132158637779.5412986042493053.43146607637414.338069621
2493487.89737641637244.3296699232494866.85439619636602.075715505
#Sta/Elev= 30
       0 1571.92    67.6 1532.85   120.4 1498.22   172.2 1455.77  217.511414.574
   258.6 1374.46  330.231369.997  523.311371.786  1001.6 1372.28 1010.571368.616
  1023.1 1362.59  1063.1 1362.14  1143.3 1362.54  1156.2 1367.17 1235.931370.653
 1337.521370.493 1542.421370.883  1685.5  1372.2  1819.4 1368.17  2035.6 1371.37
  2238.6 1367.36  2264.81369.255  2476.9 1370.06  2529.8 1388.81 2574.391392.931
    2596 1390.64  2644.6 1395.21 2780.781414.689 2883.981436.053  2953.6  1456.6
#Mann= 13 ,-1 , 0
       0      .1       0  217.51     .06       0  330.23     .05       0
  523.31     .05       0 1010.57    .045       0  1156.2      .1       0
 1235.93     .06       0 1337.52     .05       0 1542.42     .05       0
  2264.8     .05       0 2574.39     .06       0 2780.78      .1       0
 2883.98      .1       0
Bank Sta=1010.57,1156.2
XS Rating Curve= 0 ,0
Exp/Cntr(USF)=0,0
Exp/Cntr=0.3,0.1

Type RM Length L Ch R = 1 ,32016   ,543,538.4,536
XS GIS Cut Line= 4
2492713.41466667638396.6088234362493412.33808766 637936.95648351
2493626.42273913637748.0582616222494753.51546306637187.660203356
#Sta/Elev= 30
       0 1489.51   116.5 1445.35   130.9 1443.27   159.6 1426.05  176.391411.508
     217 1380.22   236.2 1379.37   250.6 1371.36   285.2 1368.83   354.6 1365.33
   563.7 1367.69  720.471365.464   899.9 1369.94   912.2 1364.92   925.1 1360.47
   999.8 1359.99  1015.8  1363.8  1095.8 1368.83 1278.141365.719    1386  1363.7
  1435.1 1368.58    1922 1365.57 2005.99  1368.8  2082.8 1388.31  2118.6  1406.8
  2167.7 1423.73 2213.951433.247  2283.7 1447.81  2355.3 1453.68  2380.8 1452.05
#Mann= 10 ,-1 , 0
       0      .1       0  176.39     .06       0   285.2     .05       0
  720.47     .06       0   899.9     .05       0   912.2    .045       0
  1015.8      .1       0 1278.14     .05       0 2005.99      .1       0
 2213.95      .1       0
Bank Sta=912.2,1015.8
XS Rating Curve= 0 ,0
Exp/Cntr(USF)=0,0
Exp/Cntr=0.3,0.1

Type RM Length L Ch R = 1 ,31478   ,622.8,659.7,704.5
XS GIS Cut Line= 4
2492940.09253294638711.4391932482493821.61756841638302.159712492
2494035.70221989638081.7784536242494728.32903347637823.617550377
#Sta/Elev= 30
       0 1414.95    20.6 1401.54    33.8 1387.34    69.1 1382.01   90.291371.206
  159.781365.392  193.451364.167  511.931363.996   698.1 1366.42  812.42 1363.76
 1028.091366.079  1048.6 1364.09  1076.8 1359.81  1134.3 1359.67    1173 1362.26
  1279.1  1364.4  1342.8 1360.41  1384.8 1364.69  1464.1 1360.95 1579.991367.251
 1665.611363.163 1681.251362.476  1709.3  1361.8  1743.4 1367.46  1781.8 1401.37
  1821.7 1428.64    1856 1449.54  1905.6  1471.9  1986.8 1494.63  2018.3 1495.02
#Mann= 12 ,-1 , 0
       0     .06       0   90.29     .05       0  159.78     .06       0
  193.45     .05       0  511.93     .05       0  812.42     .05       0
 1028.09    .025       0  1048.6    .045       0    1173      .1       0
 1579.99      .1       0 1665.61     .05       0 1681.25      .1       0
Bank Sta=1048.6,1173
XS Rating Curve= 0 ,0
Exp/Cntr(USF)=0,0
Exp/Cntr=0.3,0.1

Type RM Length L Ch R = 1 ,30818   ,492.1,496.9,499.7
XS GIS Cut Line= 4
2492883.42306637638837.3713411732494123.85472343638717.735800645
2494526.83759679638648.4731192862494929.82047015638547.727400946
#Sta/Elev= 30
       0 1440.84    43.5 1411.86   63.841393.295    87.7 1389.66   123.9 1370.82
  163.361366.458  262.881363.948  561.45 1363.08  959.531361.712 1158.581363.224
 1258.071363.196 1357.391363.216    1407 1364.44 1432.44 1359.98  1476.3 1353.97
  1537.3 1354.31 1558.541359.978  1569.8 1364.81    1586 1366.48 1655.351369.544
    1688 1371.89  1716.8 1378.29  1725.1 1384.85 1755.021424.216    1791  1455.8
  1836.4 1489.06    1923 1545.93  2017.8 1588.52 2054.021595.249  2070.5 1596.68
#Mann= 14 ,-1 , 0
       0      .1       0   63.84     .06       0  163.36     .05       0
  262.88     .05       0  561.45     .05       0  959.53     .05       0
 1158.58      .1       0 1258.07    .025       0 1357.39      .1       0
 1432.44    .045       0 1558.54      .1       0 1655.35      .1       0
 1755.02      .1       0 2054.02     .12       0
Bank Sta=1432.44,1558.54
XS Rating Curve= 0 ,0
Exp/Cntr(USF)=0,0
Exp/Cntr=0.3,0.1

Type RM Length L Ch R = 1 ,30321   ,591.2,588.6,584.7
XS GIS Cut Line= 4
2492801.56717022639435.5490438172494262.38008615639183.684747967
2494646.47313732639139.6084961932495043.15940329639051.455992646
#Sta/Elev= 30
       0 1407.25    41.61400.512   163.6 1385.67   216.3 1371.11   252.9 1366.51
   510.7 1361.26  736.841362.812   903.1 1359.04 1233.441359.082 1432.081360.796
 1531.451358.946  1579.4 1361.14 1590.341358.404  1623.7 1353.36  1728.3 1353.75
 1757.361358.402  1800.8  1366.5 1829.72 1377.34 1929.181435.213  1951.2 1447.38
  1971.7 1473.59  2003.9 1492.95 2028.661518.823  2037.4 1530.08  2086.4 1573.56
  2098.7 1590.07 2128.141611.458  2171.5 1633.16 2227.621655.315  2275.3 1665.18
#Mann= 13 ,-1 , 0
       0    .055       0    41.6     .05       0  736.84     .05       0
 1233.44     .05       0 1432.08    .025       0 1531.45     .05       0
 1590.34    .045       0 1757.36      .1       0 1829.72      .1       0
 1929.18      .1       0 2028.66     .12       0 2128.14      .1       0
 2227.62     .12       0
Bank Sta=1590.34,1757.36
XS Rating Curve= 0 ,0
Exp/Cntr(USF)=0,0
Exp/Cntr=0.3,0.1

Type RM Length L Ch R = 1 ,29732   ,600.1,598.4,594
XS GIS Cut Line= 4
2492807.86377762640014.8369242722494356.82919709639769.269235818
2494791.29510744639700.0065544592495213.16780298639592.964228723
#Sta/Elev= 30
       0 1432.42   116.3 1412.31  227.41 1398.35   278.3 1390.64  326.721388.616
   561.8 1360.81  723.981361.822   987.1  1361.3  1116.7 1354.91    1469 1360.11
 1617.821358.875  1662.9 1354.61  1707.5 1350.84  1799.1 1353.32  1799.1 1353.33
  1813.3 1355.05  1906.4 1392.42  1979.4  1416.6 2015.111437.596  2139.8 1507.24
    2181 1558.25  2193.4 1568.17 2214.511592.311  2255.3 1634.98  2292.4 1657.58
 2314.21  1676.3  2362.6 1697.77 2402.391710.387  2413.91712.933  2443.5  1719.2
#Mann= 12 ,-1 , 0
       0      .1       0  227.41     .06       0  326.72     .05       0
  723.98     .05       0 1617.82    .025       0  1662.9    .045       0
  1799.1      .1       0 2015.11      .1       0 2214.51      .1       0
 2314.21     .12       0 2402.39      .1       0  2413.9     .12       0
Bank Sta=1662.9,1799.1
XS Rating Curve= 0 ,0
Exp/Cntr(USF)=0,0
Exp/Cntr=0.3,0.1

Type RM Length L Ch R = 1 ,29134   ,532.2,517.8,495.6
XS GIS Cut Line= 4
 2493003.0586069640644.4976638962494400.90544887640373.743545858
2494784.99850004640298.1842571032495150.20172902640178.548716574
#Sta/Elev= 30
       0 1410.61   117.8 1393.19  234.921382.352  334.281373.343  433.641366.286
     5331362.536  632.361359.874   738.4 1356.75   944.9 1355.27  1186.4 1354.84
  1373.2 1357.29  1450.2 1354.01 1526.631355.462  1553.9 1354.44  1568.4 1349.92
  1632.2 1349.54  1698.8 1349.79  1717.4 1354.61 1725.371356.131  1755.9 1358.53
 1824.851391.398    1876 1411.12  1958.8 1433.03  2031.8 1461.87  2061.3 1477.73
  2103.3 1504.01  2107.8 1507.56  2117.3 1521.56  2141.2  1544.3  2199.6 1584.23
#Mann= 11 ,-1 , 0
       0     .05       0  234.92     .06       0  334.28     .05       0
  433.64     .05       0     533     .05       0  632.36     .05       0
 1526.63    .025       0  1553.9    .045       0  1717.4    .025       0
 1725.37      .1       0 1824.85      .1       0
Bank Sta=1553.9,1717.4
XS Rating Curve= 0 ,0
Exp/Cntr(USF)=0,0
Exp/Cntr=0.3,0.1

Type RM Length L Ch R = 1 ,28616   ,447.7,456.9,471.8
XS GIS Cut Line= 4
2493135.28736222641173.4126851812494533.13420419640927.844996728
2494910.93064797640751.5399896332495427.25245446 640487.08247899
#Sta/Elev= 30
       0 1413.36  188.941388.138   198.6 1385.66  288.271378.633   352.8 1375.62
   585.5  1373.1   668.4 1359.19  784.891357.733  1071.6 1356.95  1112.2 1352.84
 1182.181352.893  1281.51354.397 1482.541354.599  1553.5 1355.75  1566.7 1352.16
  1588.8 1353.12  1595.7  1350.8  1606.4 1348.32    1655 1348.06    1730 1351.35
  1774.2 1349.69  1792.21351.508  1809.6 1353.35  1916.6  1401.4  2074.3 1462.05
  2153.5 1497.55  2209.21527.232 2216.051530.562  2294.4 1571.86  2416.3 1645.71
#Mann= 12 ,-1 , 0
       0     .05       0  188.94     .06       0  288.27     .05       0
  784.89     .05       0 1182.18     .05       0  1281.5     .05       0
 1482.54    .025       0  1595.7    .045       0    1730      .1       0
  1792.2      .1       0  2209.2      .1       0 2216.05      .1       0
Bank Sta=1595.7,1730
XS Rating Curve= 0 ,0
Exp/Cntr(USF)=0,0
Exp/Cntr=0.3,0.1

Type RM Length L Ch R = 1 ,28159   ,503.2,511.4,520.1
XS GIS Cut Line= 4
2493292.70254713641658.2514546922494602.39688555641356.014299672
2495200.57458819641116.7432186152495477.62531363641003.404285482
#Sta/Elev= 30
       0 1505.43    59.6 1483.12   186.8 1423.66     232 1408.37   330.5 1397.02
   375.7 1400.48   424.9 1398.78   509.51388.391   552.2 1379.35  609.03 1372.96
   852.1 1358.09  1192.6 1352.34  1319.8 1355.01 1508.421348.192  1680.7 1354.22
  1727.9 1348.75  1849.9 1344.63  1865.3 1350.41  1891.6 1344.49 1915.52 1350.39
  1960.7 1383.63  2019.1 1407.22  2074.3 1534.54  2088.3 1545.17  2129.5 1556.67
 2147.291566.777  2215.4 1614.74  2228.4 1616.85  2241.4 1627.11  2287.7 1651.64
#Mann= 7 ,-1 , 0
       0      .1       0   509.5     .06       0  609.03     .05       0
 1508.42      .1       0  1727.9    .045       0 1915.52      .1       0
 2147.29      .1       0
Bank Sta=1727.9,1915.52
XS Rating Curve= 0 ,0
Exp/Cntr(USF)=0,0
Exp/Cntr=0.3,0.1

Type RM Length L Ch R = 1 ,27648   ,496,498,498.7
XS GIS Cut Line= 4
2493456.41433943642143.0902242032494829.07475181641758.997173032
2495395.76941748641607.8785955222495773.56586125641481.946447597
#Sta/Elev= 30
       0 1453.93    77.2 1451.66   201.8 1458.77   287.7 1456.45   376.2 1465.53
   409.5 1449.78     5271367.977   571.5 1354.58  626.941352.583   804.1 1349.31
 1026.711353.308  1182.1 1353.71  1280.8 1348.89  1493.4 1351.98 1526.291346.391
 1626.111350.237 1701.141348.148  1771.9 1348.13  1795.6  1343.5  1853.5 1342.86
  1878.4    1343 1898.221349.117    1986 1410.75  1990.1 1417.52  2005.3 1455.85
  2010.8 1463.02 2126.08 1532.85    2230 1596.21  2242.7 1600.72  2410.1 1715.72
#Mann= 10 ,-1 , 0
       0      .1       0     527     .06       0  626.94     .05       0
 1026.71     .05       0 1526.29      .1       0 1626.11    .025       0
 1701.14      .1       0  1771.9    .045       0 1898.22      .1       0
 2126.08      .1       0
Bank Sta=1771.9,1898.22
XS Rating Curve= 0 ,0
Exp/Cntr(USF)=0,0
Exp/Cntr=0.3,0.1

Type RM Length L Ch R = 1 ,27150   ,547.2,551,556.2
XS GIS Cut Line= 4
2493752.35488706642527.1832753742495049.45601068642199.759690769
2495465.03209883642105.3105798262495754.67603906642042.344505863
#Sta/Elev= 30
       0 1557.09    56.1    1547   94.76 1533.46  294.131412.033   338.2 1384.24
   374.4  1355.1  393.821351.437   419.1 1348.33   593.21350.798   819.3 1352.19
   926.6 1347.89     972 1350.41 1390.611350.344 1490.12 1351.82 1518.641347.821
  1560.6 1341.74  1609.8 1341.38    1655 1342.08  1687.41347.821  1708.3 1351.43
  1737.3 1377.17  1806.6 1419.54  1827.1 1428.54  1851.5 1487.26  1855.8 1495.14
 1888.091516.802  2003.1 1592.64  2035.9 1617.72  2048.2 1622.45  2060.4 1633.36
#Mann= 10 ,-1 , 0
       0      .1       0   94.76      .1       0  294.13     .06       0
  393.82     .05       0   593.2     .05       0 1390.61    .025       0
 1490.12      .1       0 1518.64    .045       0  1687.4      .1       0
 1888.09      .1       0
Bank Sta=1518.64,1687.4
XS Rating Curve= 0 ,0
Exp/Cntr(USF)=0,0
Exp/Cntr=0.3,0.1

Type RM Length L Ch R = 1 ,26599   ,549.2,548.1,548.1
XS GIS Cut Line= 4
2493972.73614592642980.5390079042495250.94744736642709.784889866
2495540.59138759642659.4120306962495930.98104616642546.073097563
#Sta/Elev= 30
       0  1504.9   149.2 1420.43   161.7 1419.94   198.8 1408.81   316.9 1355.12
  347.071351.994   382.3 1348.26   446.51348.613   570.4 1350.81   619.5 1345.48
   668.5 1345.26  744.791349.793  844.221349.273  1138.7 1348.48  1159.2 1343.44
 1241.94 1347.33  1374.6 1347.81  1402.3 1344.06  1416.1 1340.56  1486.9 1340.31
  1517.5 1343.78 1539.971343.947  1582.1 1343.91 1639.581378.248  1669.4 1401.16
  1689.9 1422.05  1737.9 1462.82  1823.6 1527.39 1939.751604.044  2007.1 1645.27
#Mann= 11 ,-1 , 0
       0      .1       0  347.07     .06       0   446.5     .05       0
  744.79     .05       0  844.22     .05       0 1241.94      .1       0
  1402.3    .045       0  1517.5      .1       0 1539.97      .1       0
 1639.58      .1       0 1939.75     .12       0
Bank Sta=1402.3,1517.5
XS Rating Curve= 0 ,0
Exp/Cntr(USF)=0,0
Exp/Cntr=0.3,0.1

Type RM Length L Ch R = 1 ,26051   ,565.3,562.5,562.8
XS GIS Cut Line= 4
2494205.71061958643528.3438513782495219.46441038643276.479555528
2495647.63371333643194.6236593772496050.61658669 643087.58133364
#Sta/Elev= 30
       0 1388.52    75.3 1381.97  205.071362.258  304.731355.298   427.9 1346.45
   503.9 1347.38   590.5 1343.66   697.6 1347.55  803.011345.952  1101.81344.837
 1201.151344.163  1214.9 1342.81    1276  1345.6  1284.1  1343.6  1293.4    1340
  1394.1 1339.66  1414.3 1340.51  1424.3 1343.54  1459.2 1351.39  1525.1 1377.49
  1599.11425.044  1632.7 1449.51  1636.8 1453.59  1645.1 1469.68  1649.3 1475.38
  1695.4 1511.12  1716.3 1530.45  1741.2 1550.42 1798.711586.644  1897.5 1646.22
#Mann= 10 ,-1 , 0
       0      .1       0  205.07     .06       0  304.73     .05       0
  803.01     .05       0  1101.8     .12       0 1201.15      .1       0
  1284.1    .045       0  1424.3      .1       0  1599.1      .1       0
 1798.71      .1       0
Bank Sta=1284.1,1424.3
XS Rating Curve= 0 ,0
Exp/Cntr(USF)=0,0
Exp/Cntr=0.3,0.1

Type RM Length L Ch R = 1 ,25488   ,530.9,531.2,522.6
XS GIS Cut Line= 4
2494300.15973053644126.5215540212495402.06602487643817.987791605
2495868.01497219643717.2420732652496264.70123816643603.903140133
#Sta/Elev= 30
       0 1405.58  108.231392.173   168.8 1387.35  208.171379.998   297.6 1359.66
  408.061347.315  508.011346.871   707.91346.109   819.6 1346.02   845.9 1341.31
  907.791343.246 1007.731341.808 1107.681342.563  1169.5 1340.32 1207.311343.364
  1247.3 1343.08 1306.761341.037    1366 1340.41  1492.8 1338.46  1517.4 1341.51
  1550.1 1352.13  1594.3 1373.01    1653 1413.99 1705.03  1457.5 1805.031538.396
 1905.041618.225    1965 1665.64  1981.6 1673.44 2005.041695.852  2033.6 1720.23
#Mann= 18 ,-1 , 0
       0      .1       0  108.23      .1       0  208.17      .1       0
  408.06     .06       0  508.01     .05       0   707.9     .05       0
  907.79     .05       0 1007.73     .05       0 1107.68     .05       0
 1207.31      .1       0  1247.3    .025       0 1306.76      .1       0
    1366    .045       0  1517.4      .1       0 1705.03     .12       0
 1805.03      .1       0 1905.04      .1       0 2005.04      .1       0
Bank Sta=1366,1517.4
XS Rating Curve= 0 ,0
Exp/Cntr(USF)=0,0
Exp/Cntr=0.3,0.1

Type RM Length L Ch R = 1 ,24957   ,504.8,506.1,508
XS GIS Cut Line= 4
2494533.13420419644661.7331827022495597.26085416644315.419775909
2496088.39623106 644195.784235382496396.92999348644107.631731833
#Sta/Elev= 30
       0 1406.23  148.541389.806  163.79 1387.12   264.31373.606   465.31354.407
   565.81346.537   594.8 1342.44  666.31 1342.99     889 1343.27   922.9 1336.61
  967.81 1339.19    1124 1341.12  1153.5 1338.09  1297.6 1342.94    1347 1339.82
  1372.3 1335.02  1438.5 1334.78  1454.1 1335.68 1465.551340.719 1467.241341.519
  1499.3 1352.65 1566.861393.577  1631.2 1435.56  1656.1 1465.94  1681.1 1480.19
  1766.5 1541.02  1805.9 1579.85  1868.3 1622.51  1880.8 1627.19  1945.4  1676.4
#Mann= 12 ,-1 , 0
       0      .1       0  148.54      .1       0  163.79      .1       0
   264.3      .1       0   465.3      .1       0   565.8     .06       0
  666.31     .05       0  967.81      .1       0    1347    .045       0
 1465.55      .1       0 1467.24      .1       0 1566.86      .1       0
Bank Sta=1347,1465.55
XS Rating Curve= 0 ,0
Exp/Cntr(USF)=0,0
Exp/Cntr=0.3,0.1

Type RM Length L Ch R = 1 ,24451   ,506.5,512.2,518.5
XS GIS Cut Line= 4
2494778.70189264645026.9364116852495729.48960948644793.961938024
2496151.36230503644705.8094344762496396.92999348644605.063716136
#Sta/Elev= 30
       0  1427.7    86.1 1410.44     182 1373.99     206 1367.83   373.31344.037
  376.351343.717  475.981340.838   597.2    1341   667.2 1334.26  675.24 1335.13
   691.9  1339.8   745.5  1340.7  774.871337.586   819.6 1336.62   856.7 1340.72
  1151.8 1339.69  1172.3 1334.72  1195.5 1338.27  1219.2 1337.55  1229.7 1334.49
  1311.2 1334.38    1324 1338.79  1371.81364.174 1472.791423.607  1508.7 1446.96
  1525.1 1461.39  1546.6    1470 1574.761492.084  1608.1 1509.43  1675.3 1560.92
#Mann= 11 ,-1 , 0
       0      .1       0   373.3      .1       0  376.35     .06       0
  475.98     .05       0  675.24      .1       0  774.87      .1       0
  1219.2    .045       0    1324      .1       0  1371.8     .12       0
 1472.79      .1       0 1574.76      .1       0
Bank Sta=1219.2,1324
XS Rating Curve= 0 ,0
Exp/Cntr(USF)=0,0
Exp/Cntr=0.3,0.1

Type RM Length L Ch R = 1 ,23939   ,489.1,494,500.2
XS GIS Cut Line= 4
2494929.82047015645467.6989294222495786.15907604645266.207492742
2496264.70123816645222.1312409682496466.19267484 645203.24141878
#Sta/Elev= 30
       0 1427.49   160.7 1393.25     241 1380.17   300.4 1366.87     379 1356.19
   432.4 1352.91   467.2 1343.64  496.381339.568   629.7 1340.57   654.3 1336.37
   695.51335.965   713.3 1332.98     757 1336.86   826.9 1337.78   900.4 1332.03
   996.8  1337.3  1089.2 1335.74  1145.4 1338.34  1155.4 1335.79  1161.5 1331.93
  1181.6 1331.23  1233.8 1331.79 1255.411336.667 1292.831347.162  1338.2 1371.31
  1350.3  1373.2  1366.4 1381.99  1422.6  1400.3 1491.911435.744  1562.7  1478.7
#Mann= 7 ,-1 , 0
       0      .1       0  496.38     .05       0   695.5      .1       0
  1155.4    .045       0 1255.41      .1       0 1292.83      .1       0
 1491.91      .1       0
Bank Sta=1155.4,1255.41
XS Rating Curve= 0 ,0
Exp/Cntr(USF)=0,0
Exp/Cntr=0.3,0.1

Type RM Length L Ch R = 1 ,23445   ,643.6,644.3,648.5
XS GIS Cut Line= 4
 2495187.9813734645914.7580545562495930.98104616645725.859832668
2496226.92159378645732.1564400642496510.26892661645637.707329121
#Sta/Elev= 30
       0 1395.17   262.9 1366.21     333 1355.06   353.7 1350.15   378.4 1341.87
   399.1 1337.93     428 1336.56  512.481336.888   558.3 1337.65  612.191335.532
   653.7 1333.99   679.7 1335.88   700.4 1334.21   818.4 1337.38   846.4 1334.99
   855.3 1332.45   878.4 1328.61   896.7 1328.43   950.4  1328.6   974.4 1332.06
   998.5 1335.56  1010.5 1340.42  1054.5 1342.95 1114.931353.298  1167.8 1367.77
 1215.541377.645    1288 1397.48 1316.161406.786    1345 1416.97  1361.3 1424.49
#Mann= 8 ,-1 , 0
       0      .1       0  512.48     .05       0  612.19      .1       0
   855.3    .045       0   974.4      .1       0 1114.93      .1       0
 1215.54      .1       0 1316.16      .1       0
Bank Sta=855.3,974.4
XS Rating Curve= 0 ,0
Exp/Cntr(USF)=0,0
Exp/Cntr=0.3,0.1

Type RM Length L Ch R = 1 ,22801   ,575.5,529.1,484.1
XS GIS Cut Line= 4
2495332.80334351646412.1900388592495842.82854261646355.520572293
2496220.62498638646387.0036092742496611.01464495646261.071461349
#Sta/Elev= 30
       0 1402.87   49.941394.654   151.4 1379.95   223.3 1366.05   259.5 1362.21
   295.8 1361.57   308.6 1357.22   368.2  1351.6   468.8 1345.25   513.8 1341.34
   537.2 1338.69  573.521331.599   601.4 1328.16   657.6 1328.02   749.9 1328.19
  775.131331.599   794.1 1335.51   814.1 1337.16     846 1349.61   906.8 1376.73
   919.7 1385.41   970.3 1397.23  1027.5 1406.89 1056.761414.721  1068.8 1415.73
  1091.1 1421.27  1121.5 1426.22  1171.9 1436.33  1243.6 1447.99  1302.5 1460.57
#Mann= 5 ,-1 , 0
       0      .1       0   49.94      .1       0  573.52    .045       0
  775.13      .1       0 1056.76      .1       0
Bank Sta=573.52,775.13
XS Rating Curve= 0 ,0
Exp/Cntr(USF)=0,0
Exp/Cntr=0.3,0.1

Type RM Length L Ch R = 1 ,22272   ,372.7,322.6,266.7
XS GIS Cut Line= 4
2495609.85406895 647098.520245052495905.79461657646959.994882333
2496333.96391952646771.0966604452496724.35357808 646443.67307584
#Sta/Elev= 30
       0 1433.52   190.9 1400.75   277.2 1369.01   305.7 1354.55   322.3  1351.8
   345.3 1343.16   432.7 1334.85  467.041328.705   478.1 1323.75   498.2 1323.16
   546.7 1323.17  611.751328.706   634.7 1333.21   660.1 1333.58   681.9 1339.53
   708.2  1351.3   731.8 1371.26   751.9 1385.05     765 1392.12   782.5 1398.47
   801.1 1409.87   868.9 1426.92   884.5 1438.65     895 1443.99   947.2 1453.05
     968 1451.84 1067.421462.558  1207.1 1479.84  1232.7 1481.34  1304.3 1493.86
#Mann= 4 ,-1 , 0
       0      .1       0  467.04    .045       0  611.75      .1       0
 1067.42      .1       0
Bank Sta=467.04,611.75
XS Rating Curve= 0 ,0
Exp/Cntr(USF)=0,0
Exp/Cntr=0.3,0.1

Type RM Length L Ch R = 1 ,21949   ,406.9,393.7,378.3
XS GIS Cut Line= 4
2496063.20980148647482.6132962212496157.65891242647337.791326108
2496352.85374171 646947.401667542496768.42982986646462.562898029
#Sta/Elev= 30
       0 1393.32    79.7 1382.37   147.7 1376.95   176.1 1371.68   211.9 1361.77
   237.9  1350.9   264.8 1343.53   287.9 1331.62   305.21327.529   333.9 1321.46
   404.2 1321.36  456.711327.529   477.91328.804   498.1 1332.66  521.131333.595
   542.9 1331.29   559.9 1336.87   584.3 1336.25   595.7 1343.39   646.9 1365.42
     804  1418.4   810.2 1423.29   827.4 1452.52   831.3 1456.72   841.8 1462.09
   858.1  1465.8   880.6 1464.64 1028.791480.414  1165.4 1493.48  1247.9  1505.9
#Mann= 6 ,-1 , 0
       0      .1       0   305.2    .045       0  456.71      .1       0
   477.9      .1       0  521.13      .1       0 1028.79      .1       0
Bank Sta=305.2,456.71
XS Rating Curve= 0 ,0
Exp/Cntr(USF)=0,0
Exp/Cntr=0.3,0.1

Type RM Length L Ch R = 1 ,21555   ,367.9,368.3,372.7
XS GIS Cut Line= 4
2496472.48928223647740.774199467 2496529.1587488 647602.24883675
2496642.49768193647174.0795338052496793.61625944646506.639149803
#Sta/Elev= 30
       0  1490.8    33.8 1506.02   111.6 1519.42   138.1 1530.13   147.3  1528.8
   166.8 1515.24   170.1 1508.54   176.6 1484.61   182.1 1475.59   215.9 1450.34
   231.8 1434.24   245.3 1411.37   273.1 1380.26   318.7 1346.96  369.09 1324.15
   394.1 1320.71   484.2 1320.97  502.88 1324.15  522.491326.596   542.1  1326.1
   571.1 1330.49   624.6 1344.05   858.3  1439.9   869.7 1445.38   874.7 1450.61
   895.2 1484.49  908.791487.243   993.4 1501.31 1118.571509.876  1276.9 1511.84
#Mann= 6 ,-1 , 0
       0      .1       0  369.09    .045       0  502.88    .025       0
  522.49      .1       0  908.79      .1       0 1118.57      .1       0
Bank Sta=369.09,502.88
XS Rating Curve= 0 ,0
Exp/Cntr(USF)=0,0
Exp/Cntr=0.3,0.1
